HEC-RAS study A100-00-00.prj: A100-00-00

--- A100-00-00.g01 (geometry) --- (continued)

Type RM Length L Ch R = 1 ,244940.7,697.19,1042.99,1049.47
XS GIS Cut Line= 4
     3099076.878     13779250.21     3098558.929    13777776.137
     3097259.915    13776571.441      3097247.79    13773598.166
#Sta/Elev= 30
2265.755   61.88  2929.6   62.52 2992.04   61.28 3007.94   62.91 3066.53   63.82
 3281.74    64.5 3487.05   62.29 4282.61   62.54 4760.95   61.71 4789.34   60.68
 4871.56    61.6 4920.94    60.4 4946.82   61.51 4979.34   54.31 4993.59   53.61
 5003.55   54.65 5027.86    61.5 5176.24   60.58 5403.41   62.07 5986.26   62.87
 6036.27   61.34 6096.27   62.12 6126.27   64.83 6157.06   62.78 6199.59   62.34
  6320.3   63.79 6732.83   62.99  7336.5   64.24 7482.47   63.35 8573.13   63.84
#Mann= 3 ,-1 , 0
2265.755     .07       0 4946.82     .04       0 5027.86     .07       0
#XS Ineff= 3 ,-1
2265.755 3154.72   63.51 6109.21 6124.68   63.36 6124.68 6458.63   64.15
Permanent Ineff=
       F       F       F
#Block Obstruct= 2 ,-1
 6131.42 6415.77   63.22    6495 7136.52    63.5
Bank Sta=4946.82,5027.86
XS Rating Curve= 0
Exp/Cntr=.3,.1

Type RM Length L Ch R = 1 ,243897.7,1021.54,705.99,58.86
XS GIS Cut Line= 4
     3100017.294    13779426.001     3099126.981    13777594.361
     3098323.728    13775877.606     3097478.486    13773581.687
#Sta/Elev= 30
1785.235    61.1 2709.21   60.49 2739.78   61.68 2886.96   62.67 2930.83   61.38
 3891.18   62.68  4765.6   61.61 4928.68   59.81 4958.98   60.89 4985.23   54.47
 5004.11   53.02 5044.06   60.42 5077.37   59.61 5383.32   61.83 5416.44   60.99
 5449.56   64.19 5499.24   61.375548.55561.52008 5597.37   62.55 5818.91   62.19
 5916.46   63.24 5986.36   62.33 6428.54   63.29 6543.18   62.54 6687.37   63.57
 6730.75   62.58 6885.77   64.02 7016.03   63.127143.17563.85995 8163.74   64.02
#Mann= 5 ,-1 , 0
1785.235     .07       0 4958.98     .04       0 5044.06     .07       0
5548.555     .12       07143.175     .07       0
#XS Ineff= 2 ,-1
 1785.24  3903.3    63.2 5441.41 6897.61   63.13
Permanent Ineff=
       F       F
#Block Obstruct= 1 ,-1
 5457.05 7332.33   63.17
Bank Sta=4958.98,5044.06
XS Rating Curve= 0
Exp/Cntr=.3,.1

Type RM Length L Ch R = 1 ,243191.7,393.74,102.95,34.88
XS GIS Cut Line= 6
      3100929.79    13779534.754     3100073.419    13777099.961
     3099245.585     13776229.55     3098682.899    13776204.781
     3098434.801    13775987.696     3097503.172    13773587.265
#Sta/Elev= 30
 1247.46   59.54 1385.01   60.69 2195.94   59.67 2227.75   60.79 2243.65   59.32
 2281.63   60.93 2801.68   59.97 3118.19   60.36 3149.99   61.71 4945.51   60.64
 4970.84   53.92 4984.84   53.04 4999.45    53.5 5024.85   61.14 5035.68   59.27
 5051.69   62.03 5095.76   59.42 5189.11   60.65 5654.61    60.4 5700.16   63.98
 5790.72    61.1 5888.28   61.97 6209.42   63.23 6377.27    62.1 6972.76   63.82
 7230.05   62.32 7483.56    63.4 7572.82   64.64 7947.23   63.08 8498.74   64.63
#Mann= 5 ,-1 , 0
 1247.46     .07       0 4945.51     .04       0 5024.85     .07       0
 5888.28     .12       0 7483.56     .07       0
#XS Ineff= 2 ,-1
       0    3152      64 5696.25 7334.47   63.07
Permanent Ineff=
       F       F
#Block Obstruct= 1 ,-1
 5705.33 8130.48   63.15
Bank Sta=4945.51,5024.85
XS Rating Curve= 0
Exp/Cntr=.5,.3

Type RM Length L Ch R = 1 ,243088.7,60.79,150.05,55.17
XS GIS Cut Line= 6
 3101220.584826113779229.7976261     3100326.736     13776685.21
     3099950.122    13776244.671     3098707.709     13776176.87
     3098467.319    13775967.042 3097660.725542413773931.1549715
#Sta/Elev= 30
 689.727   59.97 913.368   59.72 979.628   61.111254.194   59.06 2057.21   59.32
2421.328   61.06 2450.14   59.942571.177   60.652794.238    67.62824.961   67.01
2853.592   63.972868.808   65.072896.823   62.442910.264   63.582942.256   61.98
4477.623   60.644494.978   55.61 4499.02   53.06 4531.94   53.084532.373   54.89
4549.529   61.144559.345   59.274573.854   62.034593.675   59.865132.747   60.28
5186.772   63.92 5236.12   60.515329.425   61.696805.692    63.97719.577    64.2
#Mann= 5 ,-1 , 0
 689.727     .07       04477.623     .04       04549.529     .07       0
5329.425     .12       06805.692     .07       0
#XS Ineff= 5 ,-1
 689.7272773.575   63.412773.5754493.474    62.5    4536 5175.96    62.5
 5175.96 6732.87      64 6732.877719.577    62.5
Permanent Ineff=
       F       F       F       F       F
#Block Obstruct= 1 ,-1
 5182.63 6805.31   63.07
Bank Sta=4477.623,4549.529
XS Rating Curve= 0
Skew Angle= 25
Exp/Cntr=.5,.3

Type RM Length L Ch R = 2 ,243013  ,,,
BEGIN DESCRIPTION:
FM 2234 Rd
END DESCRIPTION:
Bridge Culvert--1,0,-1,-1, 0
Deck Dist Width WeirC Skew NumUp NumDn MinLoCord MaxHiCord MaxSubmerge Is_Ogee
25,110,2.6,25, 7, 8, , , .95, 0, 0,0,,
4006.787 4033.074463.5664463.5664599.5124599.5125184.081
    61.5    62.5    62.5    64.1    64.1    62.7    62.7
       0       0       0       0       0       0       0
 3974.16 4033.074463.5664463.5664599.5124599.5125184.0815274.711
    62.5    62.5    62.5    64.1    64.1    62.7    62.7    62.2
       0       0       0       0       0       0       0       0
BR Coef=-1 , 1 , 0 ,, 0 ,,,.8,-1,,0,
WSPro=,,,, 1 ,,,, 0 ,,,, 0 ,,,,-1 ,-1 ,-1 , 0 , 0 , 0 , 0 , 0
Multiple Barrel Culv=2,8,8,110,.012,.4,1,8,1,53.45,53.45, 3,Culvert #1  , 0 ,25
 4501.95 4490.95 4510.65 4499.65 4519.35 4508.35
Culvert Bottom n=.012
Culvert=2,8,7.6,110,.012,.4,1,8,1,53.45,4528.05,53.45,4517.05,Culvert #2  , 0 ,25
Culvert Bottom n=.012
BC Design=,, 0 ,, 0 ,,,,,,
BC HTab HWMax=67.6

Type RM Length L Ch R = 1 ,242938.7,23.56,100.84,577.87
XS GIS Cut Line= 6
 3101270.261054213779261.4389529     3100386.721    13776602.925
     3100016.263    13776147.648     3098782.913    13776076.602
     3098483.663    13775857.713 3097720.428155213773938.8351479
#Sta/Elev= 30
 634.538    59.91000.401   61.261210.229   59.021315.234   60.252231.846   59.09
2389.662   61.182575.899   60.732621.341   63.062790.767   64.192819.432   61.31
2898.309   61.082940.968   63.563928.329   59.943963.384   63.124015.958   58.88
4036.233   60.89 4468.56   60.644485.915   55.61 4488.65   53.05 4520.78   53.05
4540.466   61.144550.283   59.274564.791   62.034573.637   57.954608.304   59.23
4632.212   56.474673.059    60.35223.39261.53995 6776.5563.879837694.326   64.47
#Mann= 5 ,-1 , 0
 634.538     .07       0 4468.56     .04       04540.466     .07       0
5223.392     .12       0 6776.55     .07       0
#XS Ineff= 5 ,-1
 634.538 2784.98   63.51 2784.984483.505    62.54523.382 6307.17    62.5
 6307.17 7098.98   63.33 7098.987694.326    62.5
Permanent Ineff=
       F       F       F       F       F
#Block Obstruct= 1 ,-1
 5430.92 6927.09   63.02
Bank Sta=4468.56,4540.466
XS Rating Curve= 0
Skew Angle= 25
Exp/Cntr=.5,.3

Type RM Length L Ch R = 1 ,242837.9,52.46,617.66,984.64
XS GIS Cut Line= 6
     3101398.367    13779572.624     3100403.131    13776584.301
     3100043.784    13776111.984     3099609.393    13776094.108
     3098575.431     13774995.76     3098014.407    13773593.339
#Sta/Elev= 30
  775.13   59.93 1155.95   61.28 1397.57   58.99 2580.24   59.37 2722.53   61.43
 2880.63   60.63 2939.44   62.94 3112.35   63.98  3149.4   60.49 3298.88   62.56
 3920.27   62.33 4357.44   60.06 4401.88   62.54 4451.68   59.01  4518.3    62.6
 4853.96   63.65 4932.43   62.49 4935.28   60.14 4965.51   60.64 4990.84   53.92
 5004.84   53.04 5019.45    53.5 5044.85   61.14 5055.68   59.27 5071.69   62.03
 5140.76   60.18 5394.68    62.6 5741.33   62.15 6964.89   63.66 7972.52   64.01
#Mann= 5 ,-1 , 0
  775.13     .07       0 4965.51     .04       0 5044.85     .07       0
 5741.33     .12       0 6964.89     .07       0
#XS Ineff= 3 ,-1
  775.13 4759.95    63.2 5515.36 6125.14   62.49 6125.14 6962.46    63.4
Permanent Ineff=
       F       F       F
#Block Obstruct= 1 ,-1
 5805.77 7045.08   63.06
Bank Sta=4965.51,5044.85
XS Rating Curve= 0
Exp/Cntr=.3,.1

Type RM Length L Ch R = 1 ,242220.2,1461.62,699.21,354.17
XS GIS Cut Line= 4
     3101446.804    13779557.148     3100622.182    13777085.902
     3099664.492    13774599.267     3099243.523    13773511.241
#Sta/Elev= 30
1038.335   59.86 1216.45   59.35 1389.65   61.49 1679.65   59.38 2823.18   59.19
  2969.8   61.55 3127.93   60.45 3212.45   62.64 3317.94   61.45 3372.04   62.44
 3407.91   60.48  3609.2   62.84 4010.65   61.12  4404.1    61.7 4533.93   60.05
 4582.16   63.15  4614.3   59.63 4721.86   62.26 4901.69   63.65 4935.04   60.71
 4970.57   60.21  4992.7   53.22 5009.19   52.46 5025.85   53.23 5048.39   60.11
 5078.29   59.09 5626.06   61.66 6253.85   62.01 6419.64   63.69 7474.84   62.99
#Mann= 3 ,-1 , 0
1038.335     .07       0 4970.57     .04       0 5048.39     .07       0
#XS Ineff= 1 ,-1
 1015.93 4830.49    63.2
Permanent Ineff=
       F
#Block Obstruct= 1 ,-1
 6805.46    7562      63
Bank Sta=4970.57,5048.39
XS Rating Curve= 0
Exp/Cntr=.3,.1

Type RM Length L Ch R = 1 ,241521  ,305.52,1341.23,1587.56
XS GIS Cut Line= 5
     3102876.313    13779688.296     3101946.974    13776696.289
      3100034.18    13774816.474     3099919.113    13774510.361
     3099558.277    13773550.585
#Sta/Elev= 30
 212.255   58.57  315.54   61.12  606.57   61.44 1231.43   58.51 1343.17   61.25
 1511.83   59.07 2158.13   60.06 2189.55   58.16 2214.47   61.88 2273.25   63.04
2649.13560.17039 3136.61   61.863222.51552.26012 3333.74   50.81 3397.11   52.09
 3502.27   62.99 3624.01   58.95 3867.85   59.29 3919.75   62.574010.91560.20976
 4220.15   62.564870.98561.69989 4911.35   61.75 4927.44   59.33 4956.01   61.21
 4978.94   53.24 4995.73   52.31  5010.9    53.3 5034.57   60.34 7379.54   62.72
#Mann= 7 ,-1 , 0
 212.255     .07       02649.135     .15       03222.515     .07       0
4010.915     .15       04870.985     .07       0 4956.01     .04       0
 5034.57     .07       0
#XS Ineff= 1 ,-1
       0    4895    63.2
Permanent Ineff=
       F
#Block Obstruct= 4 ,-1
 3085.32 3485.78   60.11 3484.05 3507.24   63.31 6307.17 7217.29   62.89
 6348.74 7521.79   62.97
Bank Sta=4956.01,5034.57
XS Rating Curve= 0
Exp/Cntr=.3,.1

Type RM Length L Ch R = 1 ,240179.8,50.51,27.73,22.51
XS GIS Cut Line= 6
      3103162.04    13779687.334     3102512.254    13777579.891
     3102467.795    13777021.752     3102411.643    13776787.996
      3101992.15    13775404.188     3101168.946    13772948.093
#Sta/Elev= 30
  461.15   60.36  956.55   58.58 1007.75   61.19 1284.73   59.94 1478.65      62
 1510.05   59.14 1671.94   61.29  2192.3   59.55  2216.4   57.28 2396.26   60.12
 2497.81   58.51    2926   60.37  3489.4   59.69 3817.35   59.89 3882.69   57.94
 3914.04   62.41 3984.23   62.62 4075.96   58.94 4334.49   60.14 4404.91   60.77
 4683.43    60.9 4838.81   54.47 4885.87   54.75 4960.03   60.37 4981.37   53.45
 4990.36   52.74 5001.66   53.98 5015.54   59.53 7375.38   61.05 7503.58   63.45
#Mann= 7 ,-1 , 0
  461.15     .07       0    2926     .15       0  3489.4     .07       0
 4334.49     .15       0 4404.91     .07       0 4960.03     .04       0
 5015.54     .07       0
#XS Ineff= 1 ,-1
  327.65 3949.94      64
Permanent Ineff=
       F
Bank Sta=4960.03,5015.54
XS Rating Curve= 0
Exp/Cntr=.5,.3

Type RM Length L Ch R = 1 ,240152  ,26.42,143.57,151.64
XS GIS Cut Line= 6
 3103205.055532313779672.9902152     3102567.111    13777593.275
     3102525.721    13777083.876     3102011.161    13775397.958
      3101533.92     13774045.67     3101197.623    13772933.754
#Sta/Elev= 30
 473.685   60.09  809.56   58.45 1099.19   61.36 1373.57   58.63 1475.74   62.16
 1684.74   59.14 2338.68   59.84 2386.77   57.28 2878.08   58.64 2944.19   60.95
3221.17559.669863432.51559.11982 3886.22   58.04 3917.57   62.44 3994.37   62.42
 4027.28   57.99 4473.09   59.81 4497.15   57.75  4622.9   58.82 4638.57   61.25
 4748.29   57.63    4749    59.6    4766   54.78 4779.64   57.23 4830.77    55.7
 4950.03   60.37 4971.37    52.4  4989.4    52.4 5005.54   59.53 7518.53   61.37
#Mann= 5 ,-1 , 0
 473.685     .07       03221.175     .15       03432.515     .07       0
 4950.03     .04       0 5005.54     .07       0
#XS Ineff= 6 ,-1
  473.69    1780    63.5    4992 7518.53    62.3 3940.84    4749    61.6
  4785.8    4968    61.6    2451 3940.84    63.5    1820 2382.31    63.5
Permanent Ineff=
       F       F       F       F       F       F
#Block Obstruct= 1 ,-1
 7381.11 7699.66   62.62
Bank Sta=4950.03,5005.54
XS Rating Curve= 0
Exp/Cntr=.5,.3

Type RM Length L Ch R = 4 ,240080  ,,,
BEGIN DESCRIPTION:
Railroad
END DESCRIPTION:
Bridge Culvert--1,0,-1,-1, 0
Deck Dist Width WeirC Skew NumUp NumDn MinLoCord MaxHiCord MaxSubmerge Is_Ogee
30,70,2.6,0, 10, 10, , , .95, 0, 0,0,,
    2944    3270  4753.9  4753.9  4781.1  4781.1    4937    5063    5250    7500
    60.9    61.6    63.2    63.2    63.3    63.3    63.4    63.4    62.3    63.1
       0       0       0   60.34   60.36       0       0       0       0       0
    3229    3270  4766.9  4766.9  4794.1  4794.1    4937    5063    5250    7500
    61.5    61.6    63.2    63.2    63.3    63.3    63.4    63.4    62.3    63.1
       0       0       0   60.32   60.47       0       0       0       0       0
Pier Skew, UpSta & Num, DnSta & Num=  ,4754.5, 2 ,4767.5, 2 , 0 , 0 , 0 ,,
     1.2     1.2
       0      62
     1.2     1.2
       0      62
BR Coef=-1 , 1 , 0 ,1.25, 0 ,,,.8,0,2,0,
WSPro=,,,, 1 ,,,, 0 ,,,, 0 ,,,,-1 ,-1 ,-1 , 0 , 0 , 0 , 0 , 0
Multiple Barrel Culv=1,6,,100,.024,.9,1,2,3,52.47,52.41, 2,Culvert #1  , 0 ,30
    4976    4981    4984    4989
Culvert Bottom n=.024
BC Mult= 3 ,400,4920,400,4930
BC Mult= 2 ,4840,8000,4870,8000
BC Design=,, 0 ,, 0 ,,,,,,
BC HTab HWMax=63.07

Type RM Length L Ch R = 1 ,240008.4,21.08,41.02,29.38
XS GIS Cut Line= 6
     3103220.653    13779676.143     3102594.185    13777580.465
     3102595.469    13777009.239     3102046.295    13775159.772
     3101867.182    13774570.473      3101346.37      13772943.8
#Sta/Elev= 30
 547.535   59.78  741.81   58.46 1009.79   61.49 1444.91   58.67 1577.49   61.76
  1601.6   58.83 1769.89   58.36 2372.01   60.07 2457.35   56.77 2534.86   59.43
 2785.32   57.87 2980.32   62.02 3020.66   59.36 3165.17   61.84 3342.94   58.92
 4033.73   61.97 4249.29   58.12 4719.22   59.99  4764.9    58.8    4779   54.94
 4797.54   58.48 4828.83   56.59 4860.08   60.03 4955.03   60.37 4976.37    52.4
  4994.4    52.4 5010.54   59.53 7383.42   60.35 7483.88    63.5  7559.3   61.12
#Mann= 3 ,-1 , 0
 547.535     .07       0 4955.03     .04       0 5010.54     .07       0
#XS Ineff= 6 ,-1
  547.54    1830   62.27 3995.45    4767    61.6  4794.1    4973    61.6
    4997  7559.3    62.3    2501 3995.45   62.27    1870 2433.31   62.27
Permanent Ineff=
       F       F       F       F       F       F
#Block Obstruct= 4 ,-1
 5369.74 7690.56   61.06 5384.21 7482.71   61.25 5569.97 7526.73   60.86
 7481.23 7808.87   61.89
Bank Sta=4955.03,5010.54
XS Rating Curve= 0
Exp/Cntr=.5,.3

Type RM Length L Ch R = 1 ,239967.4,181.39,122.73,95.65
XS GIS Cut Line= 5
     3103240.091    13779680.166     3102615.027    13777576.991
     3102615.944    13777011.131     3102083.457    13775176.773
     3101388.417      13772950.7
#Sta/Elev= 30
 571.175   59.42  942.39   61.48 1133.13   58.27 1186.86   58.01 1210.74   60.77
 1234.87   58.63 1484.18   58.26 1609.37    61.6 1656.31   58.65 1718.91   60.41
 1844.09   57.26 1881.54   59.69 2055.17   60.15 2433.31   60.67 2478.73   57.58
 2532.62   60.43 2765.27    58.9  2992.4   62.72 3442.13   58.92 3603.05   61.42
 4767.49   61.19 4821.34   60.08 4852.58   55.03  4868.2   58.42  4962.1   59.64
 4986.33   52.15 5015.02   52.15 5017.07   55.68 5042.54   59.84 7573.27   61.89
#Mann= 3 ,-1 , 0
 571.175     .07       0  4962.1     .04       0 5042.54     .07       0
#XS Ineff= 8 ,-1
  571.18    1830   61.82    2501 3076.22   61.82 3076.22 3149.03    61.1
 3149.03 3995.45   61.84 3995.45 4853.85    61.1 4878.85    4980    61.1
    5019 7573.27    61.1    1870 2433.31   61.82
Permanent Ineff=
       F       F       F       F       F       F       F       F
#Block Obstruct= 2 ,-1
 5464.77 7454.31   61.37 6396.12 7711.61   61.68
Bank Sta=4962.1,5042.54
XS Rating Curve= 0
Exp/Cntr=.5,.3

Type RM Length L Ch R = 2 ,239905  ,,,
BEGIN DESCRIPTION:
FM 521 Rd
END DESCRIPTION:
Bridge Culvert--1,0,-1,-1, 0
Deck Dist Width WeirC Skew NumUp NumDn MinLoCord MaxHiCord MaxSubmerge Is_Ogee
30,75,2.6,0, 14, 14, , , .95, 0, 0,0,,
     600    1460    1831    1831    1869    1869    3360    4760    4850    4850
    5050    5050    5370    7575
    60.7    61.2    61.2    63.4    63.4    61.7    61.7    61.1    61.1    64.2
    64.2    61.1    61.1      62
       0       0       0       0       0       0       0       0       0       0
       0       0       0       0
     600    1460    1831    1831    1869    1869    3360    4760    4850    4850
    5050    5050    5370    7575
    60.7    61.2    61.2    63.4    63.4    61.7    61.7    61.1    61.1    64.2
    64.2    61.1    61.1      62
       0       0       0       0       0       0       0       0       0       0
       0       0       0       0
BR Coef=-1 , 1 , 0 ,, 0 ,,,.8,-1,,0,
WSPro=,,,, 1 ,,,, 0 ,,,, 0 ,,,,-1 ,-1 ,-1 , 0 , 0 , 0 , 0 , 0
Multiple Barrel Culv=2,2.5,5.4,45,.012,.5,1,10,1,56.38,56.38, 3,Culvert #4  , 0 ,25
  1843.5  1843.5    1850    1850  1856.5  1856.5
Culvert Bottom n=.012
Multiple Barrel Culv=1,3,,34,.024,.9,1,2,3,55.63,55.63, 2,Culvert #3  , 0 ,82.73
 2475.03 2475.03 2480.03 2480.03
Culvert Bottom n=.024
Multiple Barrel Culv=2,4,5.83,47,.012,.5,1,10,1,55.62,55.37, 3,Culvert #2  , 0 ,50
    4859    4864 4866.33 4871.33 4873.67 4878.67
Culvert Bottom n=.012
Multiple Barrel Culv=2,7,13.6,75,.012,.5,1,10,1,52.27,52.27, 2,Culvert #1  , 0 ,30
  4992.5  4957.5  5007.5  4972.5
Culvert Bottom n=.012
BC Design=,, 0 ,, 0 ,,,,,,
BC HTab HWMax=62.72

Type RM Length L Ch R = 1 ,239844.7,113.5,128.84,95.13
XS GIS Cut Line= 6
     3103428.933    13779703.063     3102767.466    13777494.109
     3102759.732    13776960.117     3102275.451    13775527.908
     3102228.575    13775368.071     3101465.198    13772860.674
#Sta/Elev= 30
  584.29   59.75  826.89   60.79  933.16   58.89 1537.93   58.58 1682.43   59.13
 1714.36   62.31 1742.67   61.89 1772.28   59.15 1970.17   56.86 2034.74   59.07
 2468.78   58.03 2570.84   60.08 2855.35   58.35 3004.28   62.08 3027.02    60.3
 3064.28   61.36  3199.3   57.23  3460.6    61.2 3597.64   58.91 3811.61   60.23
  3976.3   58.53 4406.05   62.79 4628.98   62.04 4770.25   58.23 4887.45   59.08
  4932.8   55.34 4946.73   52.15 4980.44   52.15 5038.11   59.34 7723.67   61.42
#Mann= 3 ,-1 , 0
  584.29     .07       0 4887.45     .04       0 5038.11     .07       0
#XS Ineff= 6 ,-1
  584.29    1830   61.87 2501.81 4432.31   61.87    4984 7723.67    61.1
 4432.31    4851    61.1    4885    4945    61.1    1870  2434.3   61.87
Permanent Ineff=
       F       F       F       F       F       F
#Block Obstruct= 4 ,-1
 5875.76 6556.23   60.72 7423.36 7897.44   61.46 7490.33 7827.08   60.81
       0    1710      61
Bank Sta=4887.45,5038.11
XS Rating Curve= 0
Exp/Cntr=.5,.3

Type RM Length L Ch R = 1 ,239715.9,206.16,283.02,964
XS GIS Cut Line= 6
     3103536.325    13779718.405     3102856.745    13777401.961
     3102842.788    13776978.431     3102351.814     13775504.02
      3102305.39     13775345.72      3101572.59    13772891.357
#Sta/Elev= 30
 647.195   59.86  1462.3   61.18 1802.32   58.69 1833.58   62.16 2016.77   64.31
 2190.76   61.84 2271.28   63.87 2417.92   61.49 2582.27    62.8 2630.83   56.32
 2669.44   59.02 2771.51   58.29 2787.15    60.5 2862.82   57.82 2896.57   60.75
 2959.51   57.36 3237.38   60.28 3878.13   60.43 4057.92      58 4130.14   60.62
    4216   59.04 4500.54   63.59 4642.81   62.43 4721.85   55.78 4786.28   54.89
 4879.93    55.2  4936.1    58.5 4980.36   52.74 5048.53   59.28 7765.44   61.57
#Mann= 3 ,-1 , 0
 647.195     .07       0  4936.1     .04       0 5048.53     .07       0
#XS Ineff= 2 ,-1
  364.05 2615.19   62.46 2669.44 4541.52   62.46
Permanent Ineff=
       F       F
#Block Obstruct= 3 ,-1
  436.86 1310.58   60.32  445.96    2300   61.02 6425.48 7790.67   60.85
Bank Sta=4936.1,5048.53
XS Rating Curve= 0
Exp/Cntr=.3,.1

Type RM Length L Ch R = 1 ,239432.8,56.29,967.14,1359.18
XS GIS Cut Line= 5
     3103762.591    13779765.324     3102842.137     13776692.06
     3102553.665    13775761.588     3103563.999    13774189.959
     3104009.329     13770263.67
#Sta/Elev= 30
  754.09   59.92 1323.55   59.11    1727   61.83 2007.09   58.46 2054.07   61.64
 2158.53   59.42 2727.38   60.88 2881.15   57.68 2976.35   59.08 3055.66   56.02
 3330.47   60.84    3432   58.57 4050.27   60.77 4231.36   58.04  4284.9    61.8
 4388.41   58.03 4421.93   62.11 4660.88   62.88  4718.2   62.02 4781.96   55.26
 4935.27   53.53 4942.93   53.55 4958.93   59.19 4997.49   52.32 5026.97   59.66
 8920.01   61.51  8996.7   54.33 9064.77   62.59 9150.49   60.4710756.22   61.58
#Mann= 3 ,-1 , 0
  754.09     .07       0 4958.93     .04       0 5026.97     .07       0
#XS Ineff= 3 ,-1
    6380    9060    61.2  754.09 2977.55   61.77 3133.19 4696.25   61.77
Permanent Ineff=
       F       F       F
#Block Obstruct= 7 ,-1
  573.38 1542.66   60.36  600.68 1583.62   60.86 1648.75 2035.84   60.86
 2634.81 3317.41   59.33 4675.28 4960.43   59.16 8873.72 9146.76   59.81
 9075.8410921.22   61.41
Bank Sta=4958.93,5026.97
XS Rating Curve= 0
Exp/Cntr=.3,.1

Type RM Length L Ch R = 1 ,238465.7,46.96,31.14,30.3
XS GIS Cut Line= 6
     3103832.408    13779784.711     3102957.519    13776735.275
     3103174.959    13776256.441     3103635.974    13776115.357
     3104371.653    13775579.347     3104355.941    13770196.148
#Sta/Elev= 30
 1040.64   59.71 2042.71   61.51  2399.9   58.96 3046.23   61.22 3147.56   57.37
  3413.6   59.22 3485.72   55.22 3508.87   58.27 3617.28   60.26  4471.8   60.63
 4561.61    58.2 4611.04   64.24 4643.99   65.23  4704.6   62.74 4749.18   57.83
 4922.71   56.92 4942.63   58.88 5000.59   52.12 5035.92   59.34 5129.72   58.56
 5224.94    61.5 5671.91   58.32 9392.07   59.32 9473.55   63.42 9486.49   63.16
 9517.19   56.28 9547.88   61.54 9592.92   62.38 9653.59   59.8711542.92   61.61
#Mann= 3 ,-1 , 0
 1040.64     .07       0 4942.63     .04       0 5035.92     .07       0
#XS Ineff= 4 ,-1
    5222    9460    61.1 9460.7511542.92   61.87 1040.64  3413.6   61.81
 3556.49 4641.64   61.81
Permanent Ineff=
       F       F       F       F
#Block Obstruct= 6 ,-1
  832.76 2607.51   60.99  887.37 2784.98   60.29 3030.72  3604.1   59.29
 9406.14 9651.88   59.29  9591.410652.33   60.73 10463.411606.24   61.33
Bank Sta=4942.63,5035.92
XS Rating Curve= 0
Exp/Cntr=.5,.3

Type RM Length L Ch R = 1 ,238434.6,69.89,134.09,127
XS GIS Cut Line= 6
     3103894.509    13779784.711     3103001.388      13776734.9
     3103212.418     13776269.86     3104276.163    13775775.589
     3104397.958    13775595.028      3104416.71    13770189.396
#Sta/Elev= 30
1056.785   59.49 1429.92   61.81 2355.53   58.69 2398.63    61.2 3067.15   61.21
 3178.02   57.37 3418.97   56.13 3491.47   59.18 3527.34   55.35 3593.98   59.96
 3824.08   61.17 4583.94   58.26 4669.88   65.73 4750.91   61.85 4864.47   62.81
  4910.5   57.09 4937.63   58.88 4995.59   52.12 5030.92   59.34  5095.9   59.06
 5161.13   63.97 5981.45   58.38 9271.97   59.31 9389.45   59.58 9447.65   63.38
 9467.16   60.85 9482.17   55.26 9572.18   62.05 9621.58   59.5811558.02   61.49
#Mann= 3 ,-1 , 0
1056.785     .07       0 4937.63     .04       0 5030.92     .07       0
#XS Ineff= 5 ,-1
 4750.85    4878      60    5122 5296.93      60 5296.9311558.02   61.78
 1056.79 3491.47   61.28 3593.98 4750.85   61.28
Permanent Ineff=
       F       F       F       F       F
#Block Obstruct= 6 ,-1
  764.51 2771.33   60.76  873.72 2689.42   60.26   951.9 2765.13   60.93
 3030.72 3576.79   59.23 9365.19 9651.88   59.26  9559.9 11912.4    61.1
Bank Sta=4937.63,5030.92
XS Rating Curve= 0
Exp/Cntr=.5,.3

Type RM Length L Ch R = 3 ,238367  ,,,
BEGIN DESCRIPTION:
FM 2234 Rd
END DESCRIPTION:
Bridge Culvert--1,0,-1,-1, 0
Deck Dist Width WeirC Skew NumUp NumDn MinLoCord MaxHiCord MaxSubmerge Is_Ogee
30,75,2.6,0, 10, 9, , , .95, 0, 0,0,,
    4669    4720    4870    4875    4875    5140    5140    5145    5200    5850
    65.2    65.9      68      68      68      68      68      68    65.1    61.1
       0       0       0       0    61.5    61.5       0       0       0       0
    4720    4870    4875    4875    5112    5112    5130    5200    5850
    65.9      68      68      68      68      68      68    65.1    61.1
       0       0       0    61.5    61.5       0       0       0       0
Pier Skew, UpSta & Num, DnSta & Num=  ,4940, 2 ,4925, 2 , 0 , 0 , 0 ,,
       3       3
       0      66
       3       3
       0      66
Pier Skew, UpSta & Num, DnSta & Num=  ,5030, 2 ,5015, 2 , 0 , 0 , 0 ,,
       3       3
       0      66
       3       3
       0      66
Abutment Skew #Up #Dn= , 2 , 2
    4883    4921
    61.5    58.7
    4883    4921
    61.5    58.7
Abutment Skew #Up #Dn= , 2 , 2
    5080    5130
      59    61.5
    5050    5100
      59    61.5
BR Coef=-1 , 1 , 1 ,.9, 0 ,,,.8,0,1.2,0,
WSPro=,,,, 1 ,,,, 0 ,,,, 0 ,,,,-1 ,-1 ,-1 , 0 , 0 , 0 , 0 , 0
BC Design=,, 0 ,, 0 ,,,,,,
BC HTab HWMax=65.73

Type RM Length L Ch R = 1 ,238300.5,114.48,132.36,119.2
XS GIS Cut Line= 6
     3103947.739    13779766.968     3103093.395    13776787.177
      3103268.69    13776369.615     3104326.741    13775843.147
     3104517.714    13775563.162     3104466.226    13770184.894
#Sta/Elev= 30
1119.115   59.83 2173.57   61.04 2420.29   57.09 2455.58    60.8  2496.2   57.23
  2579.1   60.63 3092.65   61.01 3170.02   59.99 3209.13    56.3 3517.87    59.1
  3570.2   55.43 3614.79   59.41 3741.48   60.77 4134.44   59.24 4355.39   61.83
  4653.4   58.36 4682.33    62.1 4819.33   64.94 4927.63   58.88 4985.59   52.12
 5020.92   59.34  5085.9   59.06 5134.18   64.08 6105.95   58.67 9341.81   59.27
 9420.03   62.68 9461.87   54.81 9514.13   62.47 9571.71    59.111579.73    61.6
#Mann= 3 ,-1 , 0
1119.115     .07       0 4927.63     .04       0 5020.92     .07       0
#XS Ineff= 5 ,-1
 5392.4911579.73    60.9    5122 5392.49      60  4737.2    4878      60
 1119.12 3517.87   60.87 3614.79  4737.2   60.87
Permanent Ineff=
       F       F       F       F       F
#Block Obstruct= 5 ,-1
  860.07 2662.12   59.91  976.35    3000   60.56 2962.46 3822.53   59.12
 9228.67 9610.92   59.15 9897.6111918.09   60.64
Bank Sta=4927.63,5020.92
XS Rating Curve= 0
Exp/Cntr=.5,.3

Type RM Length L Ch R = 1 ,238168.1,450.81,478.79,81.94
XS GIS Cut Line= 6
     3104027.583    13779749.224     3103233.623    13776820.191
     3103396.388    13776473.278     3104360.407    13775916.031
     3104596.536    13775545.155     3104529.247    13770175.891
#Sta/Elev= 30
 1229.15   59.96 1427.39   62.15 1993.41   59.05 2415.45   60.74 2540.41   57.59
 2571.65    60.7  2610.5   57.06 2634.13   59.52 2804.17   57.56  3030.3   60.25
 3608.56   58.86  3633.8   55.87 3712.01    59.2 4436.18   60.28 4539.63      60
  4945.5   61.43    4963    59.5 5005.59   52.12 5040.92   59.34 5717.73   60.16
 5870.22   57.91 6031.34   61.23 6162.09   58.38 6196.31   60.68 9244.75   59.46
 9364.78   61.88 9394.79   58.17 9444.16   63.03 9505.51   59.6811574.41   61.83
#Mann= 7 ,-1 , 0
 1229.15     .07       0 3608.56     .12       0 3712.01     .07       0
 4436.18     .12       0 4539.63     .07       0    4963     .04       0
 5040.92     .07       0
#XS Ineff= 4 ,-1
 6006.83 6020.48   60.38 6020.4811549.49   60.84 1229.15 3586.94   61.16
 3743.13 4914.68   61.16
Permanent Ineff=
       F       F       F       F
#Block Obstruct= 6 ,-1
 1032.88  2419.5   60.46 1392.49 3194.54   59.83  2408.6 2580.65   60.44
 3030.72 3781.57   59.13 9269.62 9488.05   59.48 9457.88 11732.9   60.98
Bank Sta=4963,5040.92
XS Rating Curve= 0
Exp/Cntr=.3,.1

Type RM Length L Ch R = 1 ,237689.3,896,1080.4,516
XS GIS Cut Line= 6
     3104309.063    13779734.964      3103888.75     13777398.58
     3104258.296    13776061.175     3104431.661    13775947.132
     3104683.077    13775544.867     3104614.774    13770166.889
#Sta/Elev= 30
 1635.16   60.08 2212.36   61.07 2839.15   58.13 3498.53   60.77 3631.67    59.8
 3677.39   56.44 3864.15   56.29 4004.81    59.1 4157.06   55.07  4246.2   58.59
 4564.35   58.44 4775.31   61.73 4793.33   59.05 4954.39   59.05 4989.09   51.51
 5014.45   59.19 5073.69   58.86 5752.63   60.05  5849.3   57.72 5970.37   61.15
 6102.96    58.2 6165.76    59.9 9109.47   58.92 9165.64   64.34 9207.62   54.43
 9240.66   61.43 9272.04   63.69 9315.69   59.29    9650   61.1511459.52   61.02
#Mann= 5 ,-1 , 0
 1635.16     .07       0 4004.81     .12       0 4954.39     .04       0
 5014.45     .12       0 5073.69     .07       0
#XS Ineff= 3 ,-1
 5965.87  9815.7   60.35 1635.16  4017.6   60.35 4308.44 4641.64   60.35
Permanent Ineff=
       F       F       F
#Block Obstruct= 4 ,-1
 1676.96 2062.36   60.05 2244.48 3221.14   59.93 2252.56 3235.49   59.81
 3467.58 4327.65   58.94
Bank Sta=4954.39,5014.45
XS Rating Curve= 0
Exp/Cntr=.3,.1

Type RM Length L Ch R = 1 ,236608.9,752.96,780.74,820.62
XS GIS Cut Line= 6
     3104916.719    13779717.562     3104949.202    13777038.951
     3104947.321    13776961.707     3104950.677    13776949.964
     3104949.202    13776851.731     3104703.403    13769675.945
#Sta/Elev= 30
       0   60.28  867.44   61.76 1337.52   57.68 1683.51   60.66 1905.28   59.66
 1963.98   54.29 2681.62   58.32 2712.96   58.17 2729.71   64.16 2762.92   57.39
 2781.33   52.64 2782.97    51.6 2791.63   53.74 2799.14   57.58 3165.03   58.09
 4172.25   57.64 4221.32    65.9 4299.75   60.57 4322.16   53.78    4336   57.53
 4386.19   58.84 7116.52   58.76 7204.26   61.07 7225.63    53.7 7241.93   61.28
 7297.69    61.5 8817.63   61.32 8880.08   57.66 8895.31   61.3610046.75   60.23
#Mann= 5 ,-1 , 0
       0     .07       0 2681.62     .12       0 2781.33    .041       0
 2791.63     .12       0 3165.03     .07       0
#XS Ineff= 1 ,-1
 4245.7310279.86   61.28
Permanent Ineff=
       F
#Block Obstruct= 7 ,-1
  218.43 1651.88   60.38 1795.42 2473.28      58 3975.57 4451.91   58.71
 7181.68 7309.92   59.34 7316.83 7792.46   59.82 8757.25 9032.06   60.81
Bank Sta=2762.92,2799.14
XS Rating Curve= 0
Exp/Cntr=.5,.3

Type RM Length L Ch R = 1 ,235828.2,777.47,757.49,755.61
XS GIS Cut Line= 6
     3105670.083    13780116.088     3105691.842    13777256.127
     3105703.922    13777129.468     3105703.922    13777095.916
     3105710.564     13777046.44     3105444.524    13769321.496
#Sta/Elev= 30
       0   59.38  1722.7   58.91 1778.17   55.43 2289.67   59.18 2535.64   54.55
 2597.11   57.93 2924.72   58.24 2943.64   61.07 2966.77   56.95 2991.14   53.46
 2994.58   49.69 2999.16    49.8 3007.89   56.02 3022.64   58.37 3720.47   58.16
 4901.53   59.37 4913.55   57.31 5009.25   61.65 5114.04   58.39 6998.16   58.84
 7025.04   58.65 7040.32    53.7 7058.87    53.7 7080.08   60.03 7160.37   57.37
 7277.54   59.57 8738.29   60.01 8792.39   57.66 8799.24   60.3910800.55   60.05
#Mann= 5 ,-1 , 0
       0     .07       0 2924.72     .12       0 2999.16    .041       0
 3007.89     .12       0 3720.47     .07       0
#XS Ineff= 3 ,-1
       0  1689.1    59.1 4094.92 4982.94    59.1 4982.9410800.55   60.56
Permanent Ineff=
       F       F       F
#Block Obstruct= 7 ,-1
    -121   136.1   59.56  284.69 2281.87   59.56 1703.82 2253.44   57.93
 2290.08 2711.45   57.35 6998.47 7328.24   58.55 7085.37 10841.3   59.95
 7098.7410958.45   59.85
Bank Sta=2966.77,3007.89
XS Rating Curve= 0
Exp/Cntr=.5,.3

Type RM Length L Ch R = 1 ,235070.7,512.82,609.33,655.8
XS GIS Cut Line= 6
     3106444.972    13780476.028     3106458.845    13777267.032
      3106448.78     13777198.25     3106450.457    13777164.698
     3106438.714    13777060.686     3106096.304    13768844.547
#Sta/Elev= 30
       0   59.15  318.16   60.28  330.04   56.62   639.8   60.54 2036.13   56.91
 2078.92    60.3 2113.26   55.01 2460.72   58.44 2606.81   56.76 2645.91   60.34
 2678.16    50.3 2888.79    50.3 2920.51   60.34 2949.23   57.38 3263.72   57.32
 3290.17   60.07 3312.98   56.24 3338.54   49.22 3343.96   49.45 3352.64   55.38
 3363.02    57.7 3951.25   57.44  5490.5   57.31 5611.67   61.65 5625.11   56.04
 6853.94   58.87 6918.66    53.7 6941.28   60.03 7022.35   57.3711641.81   60.24
#Mann= 5 ,-1 , 0
       0     .07       0 3263.72     .12       0 3343.96    .041       0
 3352.64     .12       0 3951.25     .07       0
#XS Ineff= 3 ,-1
       0    2786      59  3894.3 5569.97      59 5569.9711641.81   60.59
Permanent Ineff=
       F       F       F
#Block Obstruct= 6 ,-1
  -40.92  366.46   60.19 1887.02 2381.68    57.2 2564.89 2921.09   58.09
 5569.47 5697.71   58.08 6705.34 7163.36   58.37 6956.1811556.59   59.87
Bank Sta=3312.98,3352.64
XS Rating Curve= 0
Exp/Cntr=.5,.3

Type RM Length L Ch R = 1 ,234461.3,115.36,40.64,122.37
XS GIS Cut Line= 6
     3106879.311    13780580.104     3106988.291       13777282.
     3107047.685    13777124.435     3106999.763    13776926.378
      3106907.99    13772102.542     3107117.706    13768416.193
#Sta/Elev= 30
       0   59.57 2119.11   56.91 2162.43    60.3 3131.67   56.45 3154.73   59.73
 3180.79   56.68 3374.95   57.22 3391.83   53.84 3441.03   56.12 3473.03   56.61
 3504.89   49.05 3513.97   49.26 3521.34   50.82  3539.8   56.76  3593.3   59.19
 4058.41   57.15 5721.53   57.31 5845.44   61.65 5862.94   56.99 5869.11   59.64
 6859.04   58.87 6873.01   52.11 6912.15   60.03 6930.14   57.49 8524.33   57.63
 9528.17   58.82 9544.17   62.33 9565.44   59.3510269.91   58.2312196.67   60.54
#Mann= 6 ,-1 , 0
       0     .07       0 3374.95     .07       0 3441.03     .12       0
 3513.97    .041       0 3521.34     .12       0 4058.41     .07       0
#XS Ineff= 3 ,-1
       0 3468.85      59    3542  5797.5    58.9  5797.512196.67   60.72
Permanent Ineff=
       F       F       F
#Block Obstruct= 6 ,-1
 -143.67 1008.96   60.22 3368.19  3452.9    56.3 4078.62 4111.35   57.03
 6732.82 7010.69   58.18 6911.3312407.28   59.68 6912.0212343.79   59.86
Bank Sta=3473.03,3539.8
XS Rating Curve= 0
Exp/Cntr=.5,.3

Type RM Length L Ch R = 3 ,234430  ,,,
BEGIN DESCRIPTION:
Almeda School Rd.
END DESCRIPTION:
Bridge Culvert--1,0,-1,-1, 0
Deck Dist Width WeirC Skew NumUp NumDn MinLoCord MaxHiCord MaxSubmerge Is_Ogee
5,31,2.6,0, 38, 38, , , .95, 0, 0,0,,
       0     390     724    2013    2717    2982    3181    3281    3381    3457
    3458    3467    3468    3469    3492    3517    3542    3543    3544    3553
    3554    3583    3723    4064    4899    5589    5789    5889    6939    7489
    8249    8455    8692    9146   10349   11239   11649   12199
    60.2    61.2    60.8    58.6    58.9   59.37   59.28   59.34   60.33    60.3
   63.62   64.38   61.01      61   60.98   60.99      61   61.03   64.43    63.5
    60.2   60.23    58.9    59.3    58.7    59.3    60.6    59.3    59.2    58.6
    58.9    58.9    58.9    59.1    59.6    60.6    60.7      60
                                                                                
                           58.44   58.41   58.44   58.52
                                                                                
                                                                
       0     390     724    2013    2717    2982    3181    3281    3381    3483
    3484    3493    3494    3496    3519    3544    3569    3570    3571    3580
    3581    3610    3750    4091    4926    5616    5816    5916    6966    7516
    8276    8482    8719    9173   10376   11266   11676   12226
    60.2    61.2    60.8    58.6    58.9   59.37   59.28   59.34   60.33    60.3
   63.62   64.38   61.01      61   60.98   60.99      61   61.03   64.43    63.5
    60.2   60.23    58.9    59.3    58.7    59.3    60.6    59.3    59.2    58.6
    58.9    58.9    58.9    59.1    59.6    60.6    60.7      60
                                                                                
                           58.44   58.41   58.44   58.52
                                                                                
                                                                
Pier Skew, UpSta & Num, DnSta & Num=  ,3492, 2 ,3519, 2 , 0 , 0 , 0 ,,
    1.33    1.33
       0      59
    1.33    1.33
       0      59
Pier Skew, UpSta & Num, DnSta & Num=  ,3517, 2 ,3544, 2 , 0 , 0 , 0 ,,
    1.33    1.33
       0      59
    1.33    1.33
       0      59
BR Coef=-1 , 1 , 1 ,1.25, 0 ,,,.8,-1,2,0,
WSPro=,,,, 1 ,,,, 0 ,,,, 0 ,,,,-1 ,-1 ,-1 , 0 , 0 , 0 , 0 , 0
BC Design=,, 0 ,, 0 ,,,,,,
BC HTab HWMax=62.33

Type RM Length L Ch R = 1 ,234420.7,640.7,686.24,608.72
XS GIS Cut Line= 6
     3106953.876    13780591.576      3107114.48    13777259.057
     3107082.971    13777114.694     3107080.065    13774867.214
     3107011.235    13772303.296     3107243.178    13768434.118
#Sta/Elev= 30
       0   58.74     814   60.94 1511.97   58.66 1721.66   58.31 2555.15   58.22
 3103.11   56.69 3480.09   58.06 3507.04   56.86 3524.45   50.21 3540.37   49.01
 3556.51   56.79 3758.08    57.4 5727.51   56.87 5819.61   60.25 6842.96   57.88
 6862.78   52.11 6889.78    51.5 6910.87   59.44 7047.69    58.4 7061.67   54.62
 7170.93   57.76 8271.51    57.2 8392.14   57.82  8394.5    60.2  8443.8   57.66
 8469.07   60.95 8553.17   58.21 9242.91    60.8 9287.35   57.2812178.07   59.54
#Mann= 9 ,-1 , 0
       0     .07       0 1511.97     .12       0 1721.66     .07       0
 2555.15     .12       0 3103.11     .07       0 3480.09     .12       0
 3524.45    .041       0 3540.37     .12       0 3758.08     .07       0
#XS Ineff= 3 ,-1
       0 3495.84    58.6 3570.61  5797.5    58.6  5797.512178.07   59.66
Permanent Ineff=
       F       F       F
#Block Obstruct= 3 ,-1
 -107.87  492.33   59.96 6604.58 7288.55   57.71 6949.9612341.29   59.27
Bank Sta=3507.04,3556.51
XS Rating Curve= 0
Exp/Cntr=.5,.3

Type RM Length L Ch R = 1 ,233734.5,619.8,734.53,698.53
XS GIS Cut Line= 6
     3107678.896    13780600.552     3107735.504    13776956.675
      3107738.86    13776938.221     3107740.537    13776857.696
     3107735.504    13776807.368     3107385.924    13768398.977
#Sta/Elev= 30
       0   59.04  312.53   58.47  348.72    55.8  356.09   55.87  366.21   60.17
  388.99   60.55 1412.67   58.68 1715.94   58.05 3570.73   55.65  3605.5   59.99
 3660.56   58.85 3667.22    57.6 3686.25   48.01 3689.51   48.25 3698.54   49.99
 3718.37   57.19 3731.44   58.17  5759.4   56.87 5848.87   60.25 5908.12   57.88
 7028.94   57.88 7051.84   52.11 7066.24   51.47 7076.99   59.44 7126.61   61.05
 7172.21   57.58 8420.82   57.66 8433.41   60.95 8461.69   58.1512210.11   59.52
#Mann= 7 ,-1 , 0
       0     .07       0 1412.67     .12       0 1715.94     .07       0
 3660.56     .12       0 3689.51    .081       0 3698.54     .12       0
 3731.44     .07       0
#XS Ineff= 3 ,-1
       0 3299.17    58.6 3942.28 5813.42    58.6 5813.4212210.11   59.39
Permanent Ineff=
       F       F       F
#Block Obstruct= 4 ,-1
  106.87  470.23    58.7 1496.18 1859.54   58.26 6818.32 7160.31   57.16
  7125.612479.42   59.03
Bank Sta=3667.22,3718.37
XS Rating Curve= 0
Exp/Cntr=.5,.3

Type RM Length L Ch R = 1 ,232999.9,822.48,767.81,773.58
XS GIS Cut Line= 4
     3108176.993    13780334.523     3108394.804    13777142.889
     3108408.225     13777072.43     3108111.923     13768497.87
#Sta/Elev= 30
       0    57.8 1099.49      59 1414.15   58.13 2666.53   57.64 2674.55   51.26
 2702.08   48.43 2732.64   57.64 2953.34   56.33 2970.26   49.24 2989.58   49.24
 3099.51   58.94 3181.08   58.33 3205.18    56.8 3235.35   48.03 3249.89   51.05
    3260   55.71 3283.04   59.32 3532.73   56.05 5452.01   59.62 5463.05   54.63
 5557.41   60.25 5602.36   55.51 5621.52   60.25 6714.31   57.88  6727.8   51.23
 6755.66    58.4 6799.67   54.75 8121.92   56.34 8133.29    60.411850.46   59.47
#Mann= 8 ,-1 , 0
       0     .07       0 1099.49     .12       0 1414.15     .07       0
 2953.34     .12       0 3181.08     .12       0 3235.35    .041       0
 3249.89     .12       0 3532.73     .07       0
#XS Ineff= 4 ,-1
       0 2841.62    58.3    3870 5544.22    58.3 5544.2211606.83   59.19
11606.8311850.46    58.3
Permanent Ineff=
       F       F       F       F
#Block Obstruct= 7 ,-1
  -20.22  132.83   59.12  1097.8    1779   58.24 2488.13 2509.48   57.35
 2664.96 2735.09   57.09 2858.02 3096.18   56.25  6485.5 6943.51   56.87
 6756.61 11262.8    58.1
Bank Sta=3205.18,3260
XS Rating Curve= 0
Exp/Cntr=.5,.3

Type RM Length L Ch R = 1 ,232232.1,647.38,698.88,838.53
XS GIS Cut Line= 6
     3109082.625    13780011.892     3109188.312    13777082.495
      3109154.76    13776978.484      3109148.05    13776948.287
     3109136.306    13776913.057     3108970.222    13768546.711
#Sta/Elev= 30
       0   60.45 2354.18   55.94 2980.05   58.38 2994.23   54.94 3021.44   47.06
 3043.49   49.49 3051.34   55.42 3070.78   59.17 3100.44   59.29 3157.75    56.7
 5061.49   56.76 5079.72   62.65 5090.37   53.96 5113.68   62.65  5135.7   58.25
  5183.4   63.46 5231.71   51.17 5242.93   56.28  5261.5    56.8 6040.33   57.88
 6065.89   51.23 6079.82   51.26 6101.68   61.24 6118.86   58.95 6134.03   61.33
 6245.29   57.22 7751.43   55.69 7764.44   59.75 7790.86   57.1311476.66   59.47
#Mann= 5 ,-1 , 0
       0     .07       0 2967.75     .12       0 3020.08    .041       0
 3028.58     .12       0 3090.55     .07       0
#XS Ineff= 1 ,-1
 5187.7111208.19   59.29
Permanent Ineff=
       F
#Block Obstruct= 3 ,-1
 5038.17 5312.98    56.7 5917.56  6137.4   56.84 6154.5310552.02   58.98
Bank Sta=2994.23,3051.34
XS Rating Curve= 0
Exp/Cntr=.3,.1

Type RM Length L Ch R = 1 ,231533.3,699.76,655.12,619.1
XS GIS Cut Line= 6
     3109717.524    13779756.243     3109839.224    13777045.588
     3109832.513    13776980.161     3109835.869    13776919.767
     3109835.869    13776824.144     3110122.313    13768671.261
#Sta/Elev= 30
       0   57.99 2567.32   55.07 2676.28   56.01 2695.46   59.92 2711.22    60.3
 2725.89   54.44 2733.28   49.92 2734.32   47.14 2743.68   46.56 2770.88   49.05
 2791.47   56.09 2806.29    60.3 2822.56   60.89 2901.79   55.51 3652.63   56.45
 3659.66   52.43 3667.75   56.35 4776.21   55.17 4801.68   61.01 4868.78   63.04
  4911.1   55.24 7412.51   56.29  7425.1   58.35 8827.85   57.42 8895.89   57.86
 8906.43    59.8 8918.71   55.83 8937.49   58.73 9028.61   56.6911093.18   58.12
#Mann= 5 ,-1 , 0
       0     .07       0 2703.63     .12       0 2742.46    .041       0
 2750.78     .12       0 3645.22     .07       0
#XS Ineff= 1 ,-1
 4846.4211344.71    60.2
Permanent Ineff=
       F
#Block Obstruct= 3 ,-1
  128.24  329.77   57.92  3554.2 3700.76   55.24 7420.9111204.17   57.98
Bank Sta=2725.89,2791.47
XS Rating Curve= 0
Exp/Cntr=.3,.1

Type RM Length L Ch R = 1 ,230878.1,651.25,718.94,642.01
XS GIS Cut Line= 6
     3110495.964    13779444.867     3110488.458    13776944.931
      3110451.55    13776857.696     3110454.906    13776817.433
     3110449.873    13776752.007     3110713.927    13768764.674
#Sta/Elev= 30
       0   57.88    84.4   57.83   90.41    55.9   97.33   57.83  691.25   59.36
  1347.2   56.23 1785.22   56.66 1822.74    56.4 1828.58   54.44 2098.02   57.38
 2592.68   55.37  2606.4   49.57 2633.68   45.74 2651.54    54.8 2666.69   58.28
  2732.5   56.81 2752.94   54.44 3308.59   56.45 3316.28   54.58 4429.78   55.69
 4506.52   58.76 4562.45   54.36 4577.38   56.99 7066.33   56.29 7090.31   58.35
 8563.16   57.86 8587.32   56.29  8597.2   58.73  8607.3   56.6910692.88   58.12
#Mann= 5 ,-1 , 0
       0     .07       0 2532.82     .12       0 2619.33    .041       0
 2627.56     .12       0 3298.97     .07       0
#XS Ineff= 1 ,-1
 4505.1211017.06   58.23
Permanent Ineff=
       F
#Block Obstruct= 3 ,-1
  -57.39  355.91   58.51 1648.85 2015.27   55.43 7083.6510792.76   57.97
Bank Sta=2592.68,2651.54
XS Rating Curve= 0
Exp/Cntr=.3,.1

Type RM Length L Ch R = 1 ,230159.2,664.36,731.12,746.33
XS GIS Cut Line= 6
     3111118.716    13779880.793     3111120.916     13776840.92
     3111125.948    13776689.935     3111132.659    13776607.732
     3111130.981    13776555.727     3111207.689    13768855.415
#Sta/Elev= 30
       0   57.04   48.06   56.86   66.83   59.71   83.51      58  233.51   57.45
 1107.16   56.11 1433.12   58.41 2958.88   55.82    3109   55.31 3127.17   58.76
 3161.05   55.38 3185.48      46 3196.28   45.79 3226.72   55.05 3239.42   58.24
 3324.58   54.83 3695.29   56.45 3702.56   54.58 3816.98   56.19 3834.29   54.29
 4373.97   54.37 4383.87   56.19 4796.38   55.69 4830.27   57.25 4912.17   56.69
 4931.17   54.36 4947.14   56.99 8977.22   56.29 8987.55   58.7311026.19   58.12
#Mann= 5 ,-1 , 0
       0     .07       0 2958.88     .12       0 3188.66    .041       0
  3196.6     .12       0 3686.39     .07       0
#XS Ineff= 1 ,-1
 4832.7611276.45   59.16
Permanent Ineff=
       F
#Block Obstruct= 3 ,-1
  -96.22 2347.14   57.63 3774.05 4396.95   55.94 7479.7810620.31   57.82
Bank Sta=3161.05,3226.72
XS Rating Curve= 0
Exp/Cntr=.3,.1

Type RM Length L Ch R = 1 ,229428.1,325.28,315.36,312.96
XS GIS Cut Line= 6
     3111616.917    13780939.471     3111813.767    13776869.439
     3111833.899     13776805.69     3111864.096     13776693.29
     3111882.549    13776637.929      3111932.24     13768499.53
#Sta/Elev= 30
       0   57.88 3399.39   54.61  4140.3   55.36 4179.31    59.1 4182.16      56
 4199.53   45.41 4209.09   44.71  4212.1   44.29 4243.82   55.25 4283.79   58.36
 4316.32   52.01 4331.67   55.42 4719.46   55.83 4726.18   53.13 4978.98   55.84
 5157.86   60.62 5415.16   58.53 5419.46   73.14 5423.83   58.53 5700.24   54.36
 5713.04   56.99 8484.71   55.48 8505.45   58.3511172.18    56.411184.04   60.79
11196.73   58.5311203.82   52.6112388.29   52.4212418.29   57.8712454.96   58.19
#Mann= 5 ,-1 , 0
       0     .07       0 3399.39     .12       0 4199.53    .041       0
 4209.09     .12       0 4719.46     .07       0
#XS Ineff= 1 ,-1
 5160.4112428.29   59.92
Permanent Ineff=
       F
#Block Obstruct= 5 ,-1
   275.6 2808.08   57.48 5589.7410982.15   57.17 5592.84 11040.6   57.25
11065.6512428.29    57.9       0  248.78    58.7
Bank Sta=4182.16,4243.82
XS Rating Curve= 0
Exp/Cntr=.3,.1

Type RM Length L Ch R = 1 ,229112.0,40.66,39.42,39.12
XS GIS Cut Line= 6
 3111892.848534813782077.3811366 3112106.311363213779743.6033455
 3112188.253152313777813.4911553 3112107.167816313777107.2306177
 3112727.8497398 13774338.101939 3112804.652045213770376.8073489
#Sta/Elev= 30
    -353   65.53 -331.68      58 -150.44   56.71 3980.87   55.96 4933.81   54.39
 4984.47   37.88 5034.48   37.88 5090.62   56.46 5240.69   55.78 6103.81   58.37
 6182.71   57.22 6287.91   55.94 6308.95   45.53 6340.51   39.16 7293.45   37.47
 7504.54      39 7509.54   44.84 7569.55   57.53 8464.72   57.19 8554.74   43.53
 8589.74   54.69 8619.75   57.44 9454.91   58.28 9514.92   54.91 9564.93   38.84
 9667.05   38.53 9739.96   40.04 9774.97   51.94 9819.97   57.3811449.68   59.39
#Mann= 7 ,-1 , 0
    -353     .07       0 3980.87     .12       0 4933.81    .041       0
 5090.62     .12       0 5240.69     .07       0 6103.81     .12       0
 6182.71     .07       0
#XS Ineff= 3 ,-1
    -353 4815.81   57.35 5169.38 6103.81   58.57 6119.5911449.68   59.69
Permanent Ineff=
       T       T       T
#Block Obstruct= 4 ,-1
                         6272.13 7569.55   57.25 8464.72 8619.75   57.19
  9444.9 9864.98   57.81
Bank Sta=4933.81,5090.62
XS Rating Curve= 0
Exp/Cntr=.5,.3

Type RM Length L Ch R = 1 ,229073.3,165.38,165.99,167.95
XS GIS Cut Line= 6
      3111927.34     13782219.62     3112153.286     13779887.71
     3112227.535     13777957.23     3112134.723     13777251.86
     3112830.811     13774495.35     3112914.197     13770535.51
#Sta/Elev= 30
 -490.75   81.38 -406.67   80.38 -326.04   58.53 -250.44   56.68  4458.1   55.53
 4926.73   55.57 4980.42   37.91 5030.55    37.9 5090.61   57.83 5129.11   55.19
 5681.39   56.91 6062.69   61.34 6373.28   54.77 6593.67   58.59 6721.03    49.3
 6899.91   57.93 7608.38   57.69 7878.44   48.69 7973.46   55.76 8448.57   56.94
 8538.59   38.22  8603.6   56.84 8648.61      58  9483.8   57.66 9528.81   53.69
 9578.82   38.91 9753.86   38.63 9788.87   51.47 9848.88   57.78 11319.9   59.52
#Mann= 7 ,-1 , 0
 -490.75     .07       0  4458.1     .12       0 4926.73    .041       0
 5090.61     .12       0 5129.11     .07       0 5681.39     .12       0
 6062.69     .07       0
#XS Ineff= 3 ,-1
 -341.16 4880.71   57.35 5129.81 5972.08   58.57  6006.5 11319.9   61.84
Permanent Ineff=
       T       T       F
#Block Obstruct= 4 ,-1
 6593.67 6990.25   58.31 7728.41 7973.46   55.76 8448.57 8618.61   56.94
 9438.79 9848.88   57.78
Bank Sta=4926.73,5090.61
XS Rating Curve= 0
Exp/Cntr=.5,.3
